--- UB100yr2.prj (project) ---

Proj Title=Upper Brushy - 2nd run
Current Plan=p02
Default Exp/Contr=0.3,0.1
English Units
Geom File=g01
Flow File=f01
Flow File=f02
Plan File=p01
Plan File=p02
Y Axis Title=Elevation
X Axis Title(PF)=Main Channel Distance
X Axis Title(XS)=Station
BEGIN DESCRIPTION:
END DESCRIPTION:
DSS Export Rating Curves= 0
DSS Export Rating Curve Sorted= 0
DSS Export Volume Flow Curves= 0
DXF OffsetX= 0
DXF OffsetY= 0
DXF ScaleX= 1
DXF ScaleY= 10

--- UB100yr2.p02 (plan) ---

Plan Title=Hermine with dams
Program Version=4.10
Short Identifier=HermineDams
Geom File=g01
Flow File=f02
Subcritical Flow
K Sum by GR= 0
Std Step Tol= 0.01
Critical Tol= 0.01
Num of Std Step Trials= 20
Max Error Tol= 0.3
Flow Tol Ratio= 0.001
Split Flow NTrial= 30
Split Flow Tol= 0.02
Split Flow Ratio= 0.02
Log Output Level= 0
Friction Slope Method= 1
Unsteady Friction Slope Method= 2
Unsteady Bridges Friction Slope Method= 1
Parabolic Critical Depth
Global Vel Dist= 15 , 15 , 15
Global Log Level= 0
CheckData=True
Encroach Param=-1 ,0,0, 0
Computation Interval=1HOUR
Output Interval=1HOUR
Run HTab= 0
Run UNet= 0
Run PostProcess= 0
Run WQNet= 0
UNET Theta= 1
UNET Theta Warmup= 1
UNET ZTol= 0.02
UNET ZSATol= 0.05
UNET MxIter= 20
UNET MaxInSteps= 0
UNET DtIC= 0
UNET DtMin= 0
UNET MaxCRTS= 20
UNET WFStab= 2
UNET SFStab= 1
UNET WFX= 1
UNET SFX= 1
UNET DSS MLevel= 4
UNET DZMax Abort= 100
UNET Convert EG Bridges= 0
UNET Use Existing IB Tables=-1
UNET Froude Reduction=False
UNET Froude Limit= 1
UNET Froude Power= 10
UNET Time Slicing=0,0, 5
UNET Junction Losses=0
Instantaneous Interval=1HOUR
Write IC File= 0
Write IC File at Sim End=0
Echo Input=False
Echo Parameters=False
Echo Output=False
Write Detailed= 0
WQ AD Non Conservative
WQ ULTIMATE=-1
WQ Max Comp Step=1HOUR
WQ Output Interval=15MIN
WQ Output Selected Increments= 0
WQ Output face flow=0
WQ Output face velocity=0
WQ Output face area=0
WQ Output face dispersion=0
WQ Output cell volume=0
WQ Output cell surface area=0
WQ Output cell continuity=0
WQ Output cumulative cell continuity=0
WQ Output face conc=0
WQ Output face dconc_dx=0
WQ Output face courant=0
WQ Output face peclet=0
WQ Output face adv mass=0
WQ Output face disp mass=0
WQ Output cell mass=0
WQ Output cell source sink temp=0
WQ Output cell source sink nsm=0
WQ Output MaxMinRange=-1
WQ Daily Max Min Mean=-1
WQ Daily Range=0
WQ Daily Time=0
WQ Create Restart=0
WQ Fixed Restart=0
WQ System Summary=0
WQ Use Fixed Temperature=0
Sorting and Armoring Iterations= 10
XS Update Threshold= 0.02
Hydraulics Update Threshold= 0.02
Energy Slope Method= 1
Volume Change Method= 0
XS Weighting Method= 0
Number of US Weighted Cross Sections= 1
Number of DS Weighted Cross Sections= 1
Upstream XS Weight=0.25
Main XS Weight=0.5
Downstream XS Weight=0.25
Number of DS XS's Weighted with US Boundary= 1
Upstream Boundary Weight= 1
Weight of XSs Associated with US Boundary= 0
Number of US XS's Weighted with DS Boundary= 1
Downstream Boundary Weight= 0.5
Weight of XSs Associated with DS Boundary= 0.5
Sediment Output Level= 4
Mass or Volume Output= 0
Output Increment Type= 1
Profile and TS Output Increment= 10
XS Output Flag= 0
XS Output Increment= 10
Disregard all LS=0
Disregard all Conn=0
Disregard all Breaches=0
Disregard all Pumps=0

--- UB100yr2.p01 (plan) ---

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Plan Title=Simplified100Adjusted
Short Identifier=Reduced
Geom File=g01
Flow File=f01

--- UB100yr2.f02 (steady flow) ---

Flow Title=Flow for Hermine and dams
Program Version=4.10
Number of Profiles= 1
Profile Names=PF 1
River Rch & RM=Brushy,Upper           ,2840
   16300
River Rch & RM=Brushy,Lower           ,945.4837
   18800
River Rch & RM=South Brushy,Lower           ,1440
    2500
Boundary for River Rch & Prof#=Brushy,Upper           , 1
Up Type= 0
Dn Type= 0
Boundary for River Rch & Prof#=Brushy,Lower           , 1
Up Type= 0
Dn Type= 3
Dn Slope=0.008
Boundary for River Rch & Prof#=South Brushy,Lower           , 1
Up Type= 0
Dn Type= 0
DSS Import GetInterval= 0
DSS Import GetPeak= 0
DSS Import FillOption= 0

--- UB100yr2.f01 (steady flow) ---

Flow Title=Flow with dams estimated
Program Version=4.10
Number of Profiles= 1
Profile Names=PF 1
River Rch & RM=Brushy,Upper           ,2840
   16000
River Rch & RM=Brushy,Lower           ,945.4837
   24000
River Rch & RM=South Brushy,Lower           ,1440
    8000
Boundary for River Rch & Prof#=South Brushy,Lower           , 1
Up Type= 0
Dn Type= 0
Boundary for River Rch & Prof#=Brushy,Lower           , 1
Up Type= 0
Dn Type= 3
Dn Slope=0.008
Boundary for River Rch & Prof#=Brushy,Upper           , 1
Up Type= 0
Dn Type= 0
DSS Import GetInterval= 0
DSS Import GetPeak= 0
DSS Import FillOption= 0

--- UB100yr2.g01 (geometry) ---

Geom Title=FewerCS
Program Version=4.10

Junct Name=2
Junct Desc=, 0 , 0 ,-1 ,0
Up River,Reach=South Brushy    ,Lower
Up River,Reach=Brushy          ,Upper
Dn River,Reach=Brushy          ,Lower
Junc L&A=404.35,0
Junc L&A=300.27,0

River Reach=South Brushy    ,Lower
Reach XY= 29
3110007.99586976 10160928.2077233110035.5132031710160943.4711439
3110062.4229262810160949.9816296 3110091.502920610160966.0406526
3110125.3568555110161001.63080453110148.7944726910161041.9952251
 3110201.311756110161063.69662533110231.6939131910161078.8878679
 3110284.211196610161080.18970253110309.81875694 10161100.589268
3110348.2199268610161136.41629613110385.3396032810161192.6028635
3110419.6279205110161216.47453493110465.2006640110161242.9502038
3110533.7769704510161285.05084133110602.3536049410161351.8912589
 3110668.759640110161402.67232533110746.0167034310161465.6065826
 3110797.231824110161511.17932613110847.5791643610161582.7940123
3110902.2667190110161611.00589813110974.7491855910161679.5822045
 3111054.1765202 10161744.6864053111122.3187723510161813.6967657
3111185.1982397710161890.96760853111184.6926633410161890.3465468
3111269.4543048410161984.70364153111315.1763262710162019.2810002
3111354.80255935 10162036.209444

Type RM Length L Ch R = 1 ,1440    ,37.08,40.28,43.44
XS GIS Cut Line= 2
3110105.5235618710161321.39853773110479.3735359310160852.1051849
#Sta/Elev= 30
       0  767.83   31.47  769.17   34.47  768.82   51.96  774.15   70.44  775.37
   121.4  773.84  175.35  770.91  179.35  769.97  183.35  768.14  199.33  767.21
  221.82  762.59  246.29  760.05  252.79  758.32  261.28  761.41     280  760.68
  284.26  760.32  290.26  757.92  298.75  758.18     320  760.99  335.72  763.28
  343.22  763.32  354.71  764.65  370.19   771.9  384.18  780.78  401.67  789.68
  416.66  798.93  461.12  806.93  471.61  807.86  534.56  811.07     600  812.42
#Mann= 1 ,-1 , 0
       0    .045       0
Bank Sta=280,320
XS Rating Curve= 0 ,0
Exp/Cntr=0.3,0.1

Type RM Length L Ch R = 1 ,1400    ,58.34,54.87,52.52
XS GIS Cut Line= 2
3110118.1754394510161332.08289953110527.4803951110160893.3698662
#Sta/Elev= 30
       0   773.5    29.5  774.82    43.5  776.37      68  776.43    77.5  775.52
     116  774.15   145.5  771.44   176.5  770.47   190.5  766.97     204  766.03
     209  764.79   217.5  764.05     237  761.25     255  758.18  282.84  761.72
   293.5  761.08   303.5  757.91  323.39  761.03   349.5  762.82   354.5   764.3
   364.5  769.71   375.5  776.48     395  792.59   403.5  798.51     421  803.56
   436.5   805.4   471.5  808.38     528  810.43   562.5  812.35     600  812.95
#Mann= 1 ,-1 , 0
       0    .045       0
Bank Sta=282.84,323.39
XS Rating Curve= 0 ,0
Exp/Cntr=0.3,0.1

Type RM Length L Ch R = 1 ,1345.806,69.32,66.96,63.48
XS GIS Cut Line= 2
3110169.13629553 10161373.462738 3110551.948850110160928.1503084
#Sta/Elev= 30
       0  773.74  113.45  773.99  134.44  773.51  139.44  772.68  144.44  771.16
  177.92  769.14  204.41  764.75   220.9   763.1   230.9  761.18  236.39  761.32
  267.24  758.99  274.88   759.4  292.37  758.27  297.37  757.39  311.99  758.94
  339.35  762.13  352.34  767.24  372.83  779.97  387.33  792.93  401.32  801.26
  414.31  804.67  425.81  806.79  472.29  809.29  487.28  809.22  513.27   810.1
  533.76  811.87  555.25  811.98  563.25   811.2  571.75  811.14  587.24  811.97
#Mann= 1 ,-1 , 0
       0    .045       0
Bank Sta=267.24,311.99
XS Rating Curve= 0 ,0
Exp/Cntr=0.3,0.1

Type RM Length L Ch R = 1 ,1280    ,82.34,80.09,77.85
XS GIS Cut Line= 2
3110228.6453628510161449.05641893110571.46718377 10160956.640737
#Sta/Elev= 30
       0  772.97   68.44  773.64  140.38  773.61  150.87  772.34  165.36  769.85
  176.35  768.99  202.83  768.02  217.82  764.32  234.81  763.09   246.3   761.2
     280  758.97  288.76  758.34  292.26  757.46  312.24  757.13     320  757.71
  344.72  760.11  354.21  761.79  356.71  763.34   363.2  765.95  372.19  771.87
  389.18   784.7  403.17  794.02  407.66  799.63  414.66  803.58  417.66  804.37
  444.63  808.03  450.13  808.34  509.58  809.18  576.52  811.43     600  811.07
#Mann= 1 ,-1 , 0
       0    .045       0
Bank Sta=280,320
XS Rating Curve= 0 ,0
Exp/Cntr=0.3,0.1

Type RM Length L Ch R = 1 ,1200    ,66.77,70.9,75.01
XS GIS Cut Line= 2
3110311.1799746810161500.41786473110625.0966696710160989.0898191
#Sta/Elev= 30
       0  772.56   45.96   773.4  112.91  773.69   115.9  773.12  129.39  772.57
  164.86   768.4  193.84  767.78  203.83  763.99  210.83  763.81  217.82  763.07
  222.32  761.29  227.31  759.93  234.31  759.97  254.79  758.99   280.3  759.64
  303.75  758.66  314.74  758.89  320.93  759.75  332.72  760.71  343.21     763
   361.7   777.4  371.69  782.97  388.68  799.26  400.17  802.59  412.16  804.97
  437.64  807.07  463.61  808.15   478.6  808.18  513.57  809.24     600  809.48
#Mann= 1 ,-1 , 0
       0    .045       0
Bank Sta=280.3,320.93
XS Rating Curve= 0 ,0
Exp/Cntr=0.3,0.1

Type RM Length L Ch R = 1 ,1130.135,83.28,83.34,83.35
XS GIS Cut Line= 2
3110351.4279256810161511.48345943110700.3862172710161055.7543839
#Sta/Elev= 30
       0  772.82      23  773.15      99  772.81   126.5  771.04   143.5  768.29
     170  767.57   182.5  763.89     187  762.97   193.5  762.86     199  761.96
   206.5  759.87   230.5  759.24  249.49  759.37  271.18  760.14  281.49  759.62
  283.49  758.78  285.49  758.52  290.99   758.9  296.49  760.14  302.49  760.78
  304.49  761.64  311.32  762.82  320.99  766.09  336.99  777.19  353.99  787.97
  363.49  795.98  389.99  802.85  442.99  805.73  523.48  805.61  573.98  808.12
#Mann= 1 ,-1 , 0
       0    .045       0
Bank Sta=271.18,311.32
XS Rating Curve= 0 ,0
Exp/Cntr=0.3,0.1

Type RM Length L Ch R = 1 ,1047.726,87.9,87.8,87.75
XS GIS Cut Line= 2
3110413.9281287810161563.56701663110760.28209484 10161113.045936
#Sta/Elev= 30
       0   772.3   42.48  772.48  103.96   771.9  122.45   769.3  173.43  767.24
  177.43  766.76  182.43  764.48  187.42  762.85  195.92   762.1  207.92   758.8
  220.91  758.27  225.91  758.92   237.9  759.12  261.08  758.44  276.39  757.99
  283.39  759.38  301.08  760.86  307.37  761.46  321.87   766.7  338.36  783.95
  368.85  790.91  389.84  792.88  411.83     796  432.82  797.58  459.31  801.23
  513.79  800.45  518.29  800.08  543.78  803.82  558.27  804.59  568.27  804.48
#Mann= 1 ,-1 , 0
       0    .045       0
Bank Sta=261.08,301.08
XS Rating Curve= 0 ,0
Exp/Cntr=0.3,0.1

Type RM Length L Ch R = 1 ,959.9998,78.83,80.06,81.29
XS GIS Cut Line= 2
3110473.5126552610161631.02948013110837.9827268410161154.4146197
#Sta/Elev= 30
       0  771.36   64.95  771.03  103.41  770.05  129.39  770.16  137.89  769.04
  154.37  768.92  164.36  767.95  187.34  767.33  193.84   765.9  200.33  763.42
  211.32  762.46  221.82  758.56  224.31  758.04   235.3  757.23  250.29  758.33
  267.78  758.43  281.07  757.85  300.25  756.84  321.16  759.41  332.72   764.3
  334.72  764.78  344.21  769.99  350.21  772.73  372.69  780.75  408.66  785.69
  419.15  786.58   476.1  793.93  533.06  792.49  558.53   796.6     600  798.23
#Mann= 1 ,-1 , 0
       0    .045       0
Bank Sta=281.07,321.16
XS Rating Curve= 0 ,0
Exp/Cntr=0.3,0.1

Type RM Length L Ch R = 1 ,879.9999,78.36,80.11,81.85
XS GIS Cut Line= 2
3110528.6116264510161675.44671413110907.5577189310161210.2589962
#Sta/Elev= 30
       0  770.35     109  769.57     124  769.77     159  767.76     189  767.02
   192.5  766.34     200  763.32   202.5  762.85   214.5  762.31   220.5  761.02
   230.5   757.6     237  756.84     275  757.31  281.58   757.1   293.5  756.63
     309  756.54  321.61  758.82     324  759.32     329   761.7   333.5  763.17
   343.5   768.1     357  773.58     396  778.07   428.5  780.82   452.5  783.35
   473.5  784.68     532  784.27   565.5  787.34     587  788.41     600  788.58
#Mann= 1 ,-1 , 0
       0    .045       0
Bank Sta=281.58,321.61
XS Rating Curve= 0 ,0
Exp/Cntr=0.3,0.1

Type RM Length L Ch R = 1 ,800.0001,88.47,89.05,89.05
XS GIS Cut Line= 2
3110579.4402649410161718.9561415  3110978.29412610161270.7198333
#Sta/Elev= 30
       0  769.31  133.39  769.41  152.37  768.28  167.36  766.29  193.84  765.35
  205.83  762.49  223.31  761.29  256.79  757.59  266.28  756.88  278.22  757.62
  280.27  757.82  285.26  757.23  290.26  755.79  296.25  755.57  303.75  755.74
  318.31  757.49  320.73  758.06  329.72  761.49  341.22  771.05  348.21  771.74
  350.71  771.66  374.19  773.87  421.15  775.99  429.14  775.99  442.63  777.11
  530.56  777.99  567.53  777.02  576.52  777.73  586.01  779.71     600  781.63
#Mann= 1 ,-1 , 0
       0    .045       0
Bank Sta=278.22,318.31
XS Rating Curve= 0 ,0
Exp/Cntr=0.3,0.1

Type RM Length L Ch R = 1 ,712.8249,90.08,87.43,85.34
XS GIS Cut Line= 2
3110649.6051508510161761.48361553111035.8898113410161342.6468548
#Sta/Elev= 30
       0  768.69   79.47  768.32  120.95  767.68  148.44  765.36  184.93   764.7
  200.92  763.22  226.91  762.28  235.41  760.48   239.9  758.96  248.75  756.99
   253.9  756.17   258.4  756.61  273.39  755.68  289.13  756.96  307.38  759.63
  329.87  767.73  349.86  772.15  370.85  772.61  408.34  772.11  434.32  770.93
  440.32  772.49  458.31  773.29  480.31  773.51   484.8  773.43   487.8  772.92
   493.3  773.97   499.8  774.02  520.29  775.83  544.78     774  569.77  775.16
#Mann= 1 ,-1 , 0
       0    .045       0
Bank Sta=248.75,289.13
XS Rating Curve= 0 ,0
Exp/Cntr=0.3,0.1

Type RM Length L Ch R = 1 ,625.063 ,62.09,65.07,68.08
XS GIS Cut Line= 2
3110723.3897801910161833.09797363111081.4628829410161392.5598127
#Sta/Elev= 30
       0   767.1  150.42  765.39  160.92  764.87  173.41  763.33   197.4   763.5
  223.88  762.61  236.88  762.93  265.05  757.77  272.36  756.57  281.85  755.54
  305.13  755.29  307.84  755.26  332.83  760.85  351.32  767.41  364.31  766.39
   378.3   765.8   381.8  765.34  410.78  766.02  414.78  766.45  420.78   768.2
  460.26  773.73  472.75  773.81  476.75  773.42  480.25  773.65  486.74  772.57
  497.74   772.5  509.73  773.02  514.73  773.76  528.22   774.3   567.7  776.75
#Mann= 1 ,-1 , 0
       0    .045       0
Bank Sta=265.05,305.13
XS Rating Curve= 0 ,0
Exp/Cntr=0.3,0.1

Type RM Length L Ch R = 1 ,560     ,68.71,71.16,73.6
XS GIS Cut Line= 2
3110744.2781898410161874.52210343111156.6356328410161438.6765184
#Sta/Elev= 30
       0  766.27   122.9  765.82  179.35   764.9  202.83  762.57  205.83  762.74
  261.78  761.37  268.78  760.35  280.26  757.82  297.75  754.13  300.25  754.88
  304.75  754.16  320.26  755.82  327.23   756.6  333.22  756.82   361.2  766.89
   366.7   769.9  376.19  770.94  385.68  770.52  402.17  770.78  436.14  772.59
  444.13  772.36  452.13  771.34  460.62  772.87  476.11  773.95   489.6  773.95
  518.57  775.19  549.05   777.4  564.53   777.9  583.52  779.64     600  780.01
#Mann= 1 ,-1 , 0
       0    .045       0
Bank Sta=280.26,320.26
XS Rating Curve= 0 ,0
Exp/Cntr=0.3,0.1

Type RM Length L Ch R = 1 ,488.9292,81.53,84.41,87.3
XS GIS Cut Line= 2
 3110804.782990110161890.06308283111221.4498076710161499.4382078
#Sta/Elev= 30
       0  765.72  134.91  765.07   158.4  764.54  181.88     762  229.85  761.07
  237.35  760.52  241.35  759.78  253.24  756.93  258.84  755.69  268.33  754.03
  268.83  754.01  279.32  754.12  281.82  754.61   293.7  755.49  300.31  756.16
  300.81  756.36   318.3  765.77   320.8  767.49  327.79  768.71  354.28  770.26
  374.76   770.7  488.19  771.75  492.19     772  498.68  773.28  501.68  773.67
  524.17  778.29  526.67  778.58  534.66  778.55  538.66  778.44  571.14  779.34
#Mann= 1 ,-1 , 0
       0    .045       0
Bank Sta=253.24,293.7
XS Rating Curve= 0 ,0
Exp/Cntr=0.3,0.1

Type RM Length L Ch R = 1 ,404.6352,336.23,404.35,375.68
XS GIS Cut Line= 2
3110869.8871906110161918.70902283111309.9912972710161561.9380828
#Sta/Elev= 30
       0  764.97  110.41  764.93  141.89  764.64  159.87  763.21  168.37   762.2
  175.36  761.91  185.35  761.88  197.34  762.36  200.84  762.92  205.34   763.1
  207.34  763.01  208.83  763.08  222.82  761.04  227.32  760.68  230.32  759.91
  233.31  758.58  233.81  758.44   235.5  758.31  236.81  758.21  237.81  757.89
   255.3  755.12   255.8  754.97  272.78  754.54  275.99  755.54  298.76  762.61
  323.24  770.07  334.23  770.92  343.23  771.11  362.71  770.56  566.55  771.38
#Mann= 1 ,-1 , 0
       0    .045       0
Bank Sta=235.5,275.99
XS Rating Curve= 0 ,0
Exp/Cntr=0.3,0.1

River Reach=Brushy          ,Upper
Reach XY= 13
3110254.5718201710163433.03965563110286.9841569410163325.5661173
3110309.3847026810163224.46920663110356.6424821910163013.0096558
3110377.1647508410162878.77632843110429.8660890210162745.3235113
3110469.4788706910162652.89390623110553.9577043710162532.5850917
3110683.8281795110162398.8727607 3110790.560577610162323.9089998
3111082.1121598510162143.77911083111262.01173443 10162068.028278
3111354.80255935 10162036.209444

Type RM Length L Ch R = 1 ,2840    ,93.38,91.98,90.58
XS GIS Cut Line= 2
3110562.6528969410163450.49729793109988.2081796810163277.2538779
#Sta/Elev= 30
       0  777.57   38.97  775.51   43.96  777.15   48.96  778.34   63.95  778.21
   77.94  776.01   92.92   776.5  126.89  776.66  149.88  777.49  188.34   777.8
  204.83  776.22  215.32  776.08  225.31  775.36   243.3   773.2  246.79  772.28
  253.79   766.2  259.78  766.12  262.78  766.36     280  766.24     320  766.27
   361.7  766.43  412.66  768.57  425.65  768.54  431.14  768.81  435.64  768.47
  462.12  771.43   484.1  772.72  496.09  774.01  510.58  774.52     600  773.75
#Mann= 1 ,-1 , 0
       0    .045       0
Bank Sta=280,320
XS Rating Curve= 0 ,0
Exp/Cntr=0.3,0.1

Type RM Length L Ch R = 1 ,2748.022,79.66,79.68,79.68
XS GIS Cut Line= 2
3110588.5304698610163351.42498943110018.9627113610163201.1536364
#Sta/Elev= 30
       0  779.64   97.43  776.87  107.42  776.73  109.92  776.86  119.41  776.48
   129.4  775.02  146.89  774.97  149.39  775.08  157.38  774.24  162.38  774.32
  165.88  774.12  167.87   774.4  193.85  770.49  203.85  769.25  215.84  769.75
  222.33  769.66  229.83  769.92  240.82   767.8  257.31  766.44  280.22  766.31
  320.26  766.24  383.21  766.29   399.7  767.58   405.2  767.37  433.67  767.73
  437.67  768.02  449.66  769.68  499.62   774.5  518.11  773.87  589.06  773.52
#Mann= 1 ,-1 , 0
       0    .045       0
Bank Sta=280.22,320.26
XS Rating Curve= 0 ,0
Exp/Cntr=0.3,0.1

Type RM Length L Ch R = 1 ,2668.501,42.69,43.9,45.11
XS GIS Cut Line= 2
3110605.7472989310163273.8585435 3110034.587680110163123.0287927
#Sta/Elev= 24
       0  779.48  161.93  776.64  173.92  775.92  204.91  771.89  208.41  771.71
  208.91  771.65   217.9  769.53   231.9   767.2   235.4  766.39  275.96  766.27
  294.37  766.21  295.87  766.05  296.37  766.04  299.37  766.18  316.13  766.13
  355.84  766.31  380.83  766.75  430.31   768.2  433.81  768.49  438.31  769.52
  474.29  774.05  517.78  773.17  577.75  773.19  590.74  772.96
#Mann= 1 ,-1 , 0
       0    .045       0
Bank Sta=275.96,316.13
XS Rating Curve= 0 ,0
Exp/Cntr=0.3,0.1

Type RM Length L Ch R = 1 ,2624.488,62.49,60.37,58.25
Node Name=USDamonBC
XS GIS Cut Line= 2
3110600.5599733610163235.87600793110038.0601141210163069.2093465
#Sta/Elev= 30
       0  779.42  143.42  776.64   180.9  772.28   185.9  770.58  199.39   763.8
  205.38  762.08  214.38   761.2  219.38  758.96  232.87  758.12  243.86  758.09
  259.07  759.26  262.35  759.28  273.35   757.6  279.34  758.54  284.84  757.95
  293.34  758.67  299.38  758.34  307.33  758.02  312.83  758.71  320.32  758.75
  328.32  758.04  345.81  759.83   352.3  759.99   359.8  762.02  376.29  762.96
  391.28  766.38  423.76   771.2  435.26  771.37  451.25  773.11  586.67  772.43
#Mann= 1 ,-1 , 0
       0    .045       0
Bank Sta=259.07,299.38
XS Rating Curve= 0 ,0
Exp/Cntr=0.3,0.1

Type RM Length L Ch R = 1 ,2564.688,45.46,44.83,44.2
XS GIS Cut Line= 2
3110624.86569902 10163164.6953763110046.3645594410163025.8852862
#Sta/Elev= 30
       0  779.15    27.5  779.09   47.49  778.22  118.48  776.68  128.48  776.69
  139.48  775.67  163.98  772.51  168.48  771.74  173.48  770.33  182.98  766.62
  206.97  758.36  207.97  758.11  217.97  756.92  221.97  756.79  270.11  756.63
  285.96  756.43  289.96  757.43  290.96  756.68  291.46  756.41  305.96  756.35
  310.21  756.47  312.46  756.33  345.45  757.79  356.95  758.74  364.45  760.06
  391.45  766.18  421.44   770.6  475.44  772.77  562.43  772.57  594.92  771.85
#Mann= 1 ,-1 , 0
       0    .045       0
Bank Sta=270.11,310.21
XS Rating Curve= 0 ,0
Exp/Cntr=0.3,0.1

Type RM Length L Ch R = 1 ,2520    ,40.06,40.06,40.21
XS GIS Cut Line= 2
3110640.6438826910163117.71056193110055.0886233410162986.8482908
#Sta/Elev= 30
       0  778.93     116  776.58   169.5  770.05     179  767.99     184  764.44
     193  760.17   202.5  758.72   208.5  758.48     221  758.78   224.5  758.66
     228  758.08   243.5  757.23     266  757.33     273  756.51  277.73   756.5
     294  756.17   297.5  756.65     299  756.22  317.79  757.41     345  759.04
     353  759.16     377  765.33   406.5  769.56   428.5  770.82     439  771.78
     450  773.29   458.5  773.62   483.5  772.75     547  772.45     600   771.6
#Mann= 1 ,-1 , 0
       0    .045       0
Bank Sta=277.73,317.79
XS Rating Curve= 0 ,0
Exp/Cntr=0.3,0.1

Type RM Length L Ch R = 1 ,2480    ,98.43,97.93,97.28
XS GIS Cut Line= 2
3110649.3682746910163078.67356643110063.8126872810162947.8112953
#Sta/Elev= 30
       0  778.17   117.9  775.59  125.89  773.85  130.39  773.53  161.87  768.88
  173.86  764.72  184.85  760.52  188.84  759.68  193.34   758.4  279.96  756.15
  293.26  755.29  299.25  755.93  319.23  757.49  320.51  757.72  331.72  758.42
  336.72  759.04  346.71  760.92  349.21  761.83   357.7  763.68  387.18   767.3
  409.16  770.59  419.15  770.67  420.65  770.57  437.63   772.7  440.63  772.87
  442.63   772.8  460.12  773.56   474.6  772.52  540.55  772.49     600  771.41
#Mann= 1 ,-1 , 0
       0    .045       0
Bank Sta=279.96,320.51
XS Rating Curve= 0 ,0
Exp/Cntr=0.3,0.1

Type RM Length L Ch R = 1 ,2384.113,67.56,73.33,79.1
XS GIS Cut Line= 2
3110665.25111693 10162979.5028333110093.6154491910162860.8757737
#Sta/Elev= 30
       0  777.07   31.99   776.5   77.48  776.57   94.47  776.26  101.47  775.68
  105.47  776.15  112.46  775.89  124.46  774.71  128.46  772.82  132.96  769.68
  140.46  765.46  144.45  764.41  178.44   763.2  191.94  757.75  193.94  757.43
  247.42  756.91  289.19  755.52   305.4  754.61   309.4  754.88   312.9   754.3
   322.9  754.67  329.78  757.27  349.89  765.04  372.88  770.06  408.37  772.21
  420.87  772.46  448.86  772.37  455.86  771.87  509.84  772.01  583.82  770.92
#Mann= 1 ,-1 , 0
       0    .045       0
Bank Sta=289.19,329.78
XS Rating Curve= 0 ,0
Exp/Cntr=0.3,0.1

Type RM Length L Ch R = 1 ,2311.327,70.17,71.33,72.48
XS GIS Cut Line= 2
3110668.2681712810162949.41759133110106.9379290910162746.2923414
#Sta/Elev= 30
       0  776.95   61.99  776.06   67.99  775.32   70.99  775.62   77.49  775.11
   91.99  775.25   99.99   774.8  102.99     774  114.99  768.76  123.49  766.55
  127.99  764.76  134.49  763.92  143.49  764.59  154.49  764.15  166.99  763.06
  176.99  758.09  181.49  757.07  227.98  757.24  276.82  755.78  301.98  753.82
  314.48  754.67  316.83  755.53  321.97  758.03  331.97  765.41  343.97  767.19
  355.47  769.83  374.97  769.73  393.47  771.98  486.96   771.5  596.95  769.93
#Mann= 1 ,-1 , 0
       0    .045       0
Bank Sta=276.82,316.83
XS Rating Curve= 0 ,0
Exp/Cntr=0.3,0.1

Type RM Length L Ch R = 1 ,2240    ,78.85,80,81.15
XS GIS Cut Line= 2
3110694.3829484310162892.26580283110136.3223847710162671.8843538
#Sta/Elev= 30
       0  776.47      47  775.46    52.5  775.68      59  775.07      77  771.89
      95  768.23   121.5  764.23   135.5  763.87     142  763.37     156     761
     162  759.62   251.5  755.96   257.5  755.34   266.5   755.5   268.5  755.37
     280     755   291.5  754.38   297.5  753.81     303  754.47   309.5  754.67
     310  754.78     320  758.22   341.5  765.64     351  767.55   364.5  769.21
   376.5  770.32     406  771.98   422.5  771.55     545  770.41     600  769.48
#Mann= 1 ,-1 , 0
       0    .045       0
Bank Sta=280,320
XS Rating Curve= 0 ,0
Exp/Cntr=0.3,0.1

Type RM Length L Ch R = 1 ,2160    ,72.75,76.49,80.23
XS GIS Cut Line= 2
3110721.55809093 10162826.2866043110170.0710049310162589.9343864
#Sta/Elev= 30
       0  775.62   47.96  774.71   49.96  774.79   52.96  774.45   65.45  771.41
   80.93   769.2   84.93  768.36   92.42  767.21  102.91  766.51   121.4  764.79
  137.39  763.95  165.36  760.12  185.35  758.68     280  755.11  286.26  754.71
  289.26  754.15  300.25  753.48  315.74  753.97  316.24  754.05     320  755.41
  330.23  759.37  336.22  762.28  341.22  765.03  344.71  766.14  352.21  767.81
  352.71  767.89   357.7  767.87   366.2  768.47  393.67  771.43     600  768.42
#Mann= 1 ,-1 , 0
       0    .045       0
Bank Sta=280,320
XS Rating Curve= 0 ,0
Exp/Cntr=0.3,0.1

Type RM Length L Ch R = 1 ,2083.508,78.93,83.51,88.09
XS GIS Cut Line= 2
3110735.97669727 10162779.2788243110222.0876331910162499.7646193
#Sta/Elev= 30
       0  774.14      21  773.97    28.5  773.76    81.5  767.24   103.5  765.39
     152  762.28   156.5  761.65   161.5  760.45   168.5  759.44     181  758.51
   218.5  757.92  272.49   756.1  275.99  755.88  279.49  755.12  283.49  753.62
  285.99   753.3  291.49  753.07  303.99  752.98  304.99  753.23  307.49  754.63
  312.76   757.2  331.99   766.1  339.99  766.79  352.49  766.95  371.49  770.73
  375.49  771.25  408.49  770.94  455.49  771.17  524.49  769.62  584.99  767.03
#Mann= 1 ,-1 , 0
       0    .045       0
Bank Sta=272.49,312.76
XS Rating Curve= 0 ,0
Exp/Cntr=0.3,0.1

Type RM Length L Ch R = 1 ,2000    ,75.15,78.43,81.71
XS GIS Cut Line= 2
3110772.4198658510162743.51347563110281.3850867710162398.7169211
#Sta/Elev= 29
       0  773.66      30  773.21    45.5  772.01      93   766.5     173  761.31
   199.5  758.37     220   757.5     280  755.89     286  755.74     295  754.66
   299.5  753.72   300.5   753.4     307  752.54   307.5  752.51   316.5  753.07
   318.5  753.07     319   753.2     320  753.58     344  762.48   348.5  764.29
     350  764.73     352  765.05   366.5  765.93   381.5  768.77   394.5  770.35
     441  770.78   541.5  769.74   569.5  768.85     600  766.73
#Mann= 1 ,-1 , 0
       0    .045       0
Bank Sta=280,320
XS Rating Curve= 0 ,0
Exp/Cntr=0.3,0.1

Type RM Length L Ch R = 1 ,1921.568,78.49,81.57,84.65
XS GIS Cut Line= 2
3110805.4211121810162701.15365223110350.56014526 10162322.681312
#Sta/Elev= 30
       0   773.2   31.99   772.7   56.97  770.65   83.96  767.54  120.44  764.88
  135.44  764.09  149.43  762.61  155.43  762.59  187.41  760.84  191.41  760.87
  193.91  760.62  201.41  758.64   208.4  757.33  278.65  755.59  296.86  754.98
  298.86  753.81  301.36  754.85  304.36  754.75  312.36  753.15  317.85  752.91
  318.77  752.94  324.35  753.18  349.34  762.43  357.33   763.5  363.33  765.23
  382.32  766.93   436.3  770.72  483.78  770.67  536.75  769.88  591.73  768.01
#Mann= 1 ,-1 , 0
       0    .045       0
Bank Sta=278.65,318.77
XS Rating Curve= 0 ,0
Exp/Cntr=0.3,0.1

Type RM Length L Ch R = 1 ,1840    ,95.92,100.9,105.89
XS GIS Cut Line= 2
3110847.8327727610162660.60156793110417.4307464410162242.5656586
#Sta/Elev= 30
       0   772.6    60.5  770.84     166   762.7   233.5   756.6     249  756.09
     280  755.57     291  755.07   294.5  755.12     296  754.99   299.5  753.46
     300  753.49   300.5  754.37     301  754.81     303  754.53     308  752.98
     315  752.25     320  752.84     325  752.79   339.5  758.73   340.5  759.03
     362  763.18   386.5  765.43     390  765.53   411.5  770.48   426.5  771.45
     441     771   449.5  770.58     536  770.04     567  768.71     600  766.86
#Mann= 1 ,-1 , 0
       0    .045       0
Bank Sta=280,320
XS Rating Curve= 0 ,0
Exp/Cntr=0.3,0.1

Type RM Length L Ch R = 1 ,1739.096,56.55,59.1,61.64
XS GIS Cut Line= 2
3110894.3218530110162617.63380613110524.1710185110162156.0146506
#Sta/Elev= 30
       0  772.08   74.96  770.73   83.46  770.25   92.95  769.36   99.45  768.27
  118.44   767.2  131.93  765.75  252.87  755.71  280.57  755.12  285.35  754.97
  292.85   753.2  316.84  752.83  320.65   753.6  325.33   754.7  336.83  758.35
  368.31  762.91  374.81  763.37   379.3  763.01   390.8  763.19   395.3  764.43
  403.79  767.54  408.29  768.73  413.79  769.11  416.29  769.47  436.28  769.91
  440.27  769.55  448.27  770.12  456.27  770.07  464.26  769.66   591.7  767.19
#Mann= 1 ,-1 , 0
       0    .045       0
Bank Sta=280.57,320.65
XS Rating Curve= 0 ,0
Exp/Cntr=0.3,0.1

Type RM Length L Ch R = 1 ,1680    ,77.64,80,82.36
XS GIS Cut Line= 2
 3110927.054727210162594.6436946 3110582.202726610162103.6479574
#Sta/Elev= 30
       0   771.8      61   771.1    81.5   770.6     106  768.87     141  765.51
     216  760.15   229.5  758.66     251  755.12     253  754.95     280  755.11
   286.5  755.32     289  755.23     295  754.05     300  753.94   306.5  752.75
     320  752.95   328.5  752.87   330.5  753.58     337  756.61     344  760.18
     351  761.47   362.5  761.27     374  762.63   389.5  762.24     401  762.53
   433.5  764.38     448  764.93     490  767.25     544  767.84     600  765.73
#Mann= 1 ,-1 , 0
       0    .045       0
Bank Sta=280,320
XS Rating Curve= 0 ,0
Exp/Cntr=0.3,0.1

Type RM Length L Ch R = 1 ,1600    ,80,80,80
XS GIS Cut Line= 2
3110978.9463556710162560.15754313110663.5821570210162049.7208999
#Sta/Elev= 30
       0  771.64   116.9   769.1  134.39  767.87  164.86  767.12  186.84  762.36
  200.83  760.06  208.83  760.04  217.82  758.75  224.81   758.9  261.78  755.05
  271.77  754.43     280  755.04  299.75  754.31  301.25  754.76  314.24  752.51
     320  752.67  323.73  752.53  344.71  754.53  375.69  760.15  398.67  762.53
  407.66  762.14  432.64  765.21  443.13  765.76   475.1  765.69   482.6  765.18
  488.59  763.47  496.59  762.45  547.04  765.65  576.02  764.97     600  763.35
#Mann= 1 ,-1 , 0
       0    .045       0
Bank Sta=280,320
XS Rating Curve= 0 ,0
Exp/Cntr=0.3,0.1

Type RM Length L Ch R = 1 ,1520    ,79.65,79.69,79.73
Node Name=J365
XS GIS Cut Line= 2
3111047.0046185310162518.10907083110731.6404198410162007.6724276
#Sta/Elev= 30
       0  771.44   26.98  770.64   38.47  769.92   44.96   770.1  147.88  767.65
  196.84  763.51  216.82  760.89  223.81  759.58  265.78  758.03     280  756.98
  285.26  756.22  289.76  754.82  311.24  752.59     320  753.93   357.2  759.77
  366.69  760.69  378.68  760.16  388.18  760.52  428.64   763.9  455.62  768.66
  502.58  768.57  520.07  767.37  528.06  767.54  546.04  762.34  552.04  761.79
  556.04  762.07  572.52  765.02  585.01  765.43   595.5  764.77     600   764.9
#Mann= 1 ,-1 , 0
       0    .045       0
Bank Sta=280,320
XS Rating Curve= 0 ,0
Exp/Cntr=0.3,0.1

Type RM Length L Ch R = 1 ,1440.313,78.06,77.66,77.27
XS GIS Cut Line= 2
3111127.26561284 10162497.051042 3110799.698682710161965.6239553
#Sta/Elev= 30
       0  771.85   23.49  771.62   29.49  771.64  220.42  764.89  252.91  762.21
   285.9  758.16  294.89  757.48  304.27  756.34  314.88  754.55  318.88  753.53
  323.88  753.37  324.38  753.27  325.38  752.67  325.88   752.5  340.88  752.48
  344.27   753.1  351.37  754.46  362.87  756.25  372.36  758.49  389.36  759.78
  401.85  760.27  403.35  760.51  418.35  761.28  420.35  761.55  473.83  765.68
  485.32  765.95  487.32  766.52  492.82  767.41  591.79  766.56  624.28  765.58
#Mann= 1 ,-1 , 0
       0    .045       0
Bank Sta=304.27,344.27
XS Rating Curve= 0 ,0
Exp/Cntr=0.3,0.1

Type RM Length L Ch R = 1 ,1362.649,74.45,73.7,72.94
XS GIS Cut Line= 3
3111188.0295989210162477.51991313111131.3338461810162351.8233141
 3110873.129310110161942.0390287
#Sta/Elev= 30
       0  771.08   76.44  768.92  146.89  767.65  251.36  764.76  276.35   762.3
  320.76  755.85  326.83  755.14  336.83  752.92  347.83  752.65  353.82  752.87
  360.76   753.9  370.32  755.35  382.82  757.75  399.81  759.07  409.81  759.26
   417.3   758.9   426.3  760.47   434.3     761  451.29  763.61  461.29  764.71
  465.29  764.54  479.79  766.58  486.78  766.62  493.78  765.81  499.78  765.52
  512.28  763.94  518.27  764.45  544.27  765.21  596.25   764.3  622.24   764.5
#Mann= 1 ,-1 , 0
       0    .045       0
Bank Sta=320.76,360.76
XS Rating Curve= 0 ,0
Exp/Cntr=0.3,0.1

Type RM Length L Ch R = 1 ,1288.952,42.84,43.19,42.91
XS GIS Cut Line= 3
3111255.3040706810162475.34964183111184.1959451710162291.8693658
3110949.3141970910161932.8149658
#Sta/Elev= 30
       0  770.82  145.84  767.63  227.75  766.07  229.74  765.76  251.72  766.01
  256.72  765.86   273.2  764.06  304.67  762.65  318.65  760.19  324.15  759.68
  345.12  755.71  355.46  754.52  372.59  752.49  389.08  752.65  396.12  753.39
  419.05  755.27  428.04  757.99  448.52  759.02  453.01  758.98  455.01   758.6
  456.51  758.59     464  759.55     467  759.55  488.97  761.06  494.47  761.18
  498.46   761.7  519.94   762.1  545.91  763.21  582.38  764.15  625.83  764.45
#Mann= 1 ,-1 , 0
       0    .045       0
Bank Sta=355.46,396.12
XS Rating Curve= 0 ,0
Exp/Cntr=0.3,0.1

Type RM Length L Ch R = 1 ,1245.758,273.89,300.27,329.17
XS GIS Cut Line= 3
3111290.2433052710162437.80640993111223.6105645310162277.3759564
3110992.7169974410161917.6240513
#Sta/Elev= 30
       0  770.25  227.21  765.64  244.21  764.89  268.71  763.27  289.71  761.25
  321.71  755.84  326.71  755.16  334.12  754.48  354.21  752.38  355.71  752.57
  374.72  752.88  380.21  753.73  391.71  754.08  392.21  754.19  398.71  756.95
  399.21  757.06   403.7  757.46   405.7  757.46   431.2  759.58   434.7  759.64
   454.7  761.25   472.7  761.71   482.2  762.27   502.2  764.25   517.2  764.57
   544.7  764.07   551.7  764.32  557.19  764.84  565.69  765.12  601.19  765.04
#Mann= 1 ,-1 , 0
       0    .045       0
Bank Sta=334.12,374.72
XS Rating Curve= 0 ,0
Exp/Cntr=0.3,0.1

River Reach=Brushy          ,Lower
Reach XY= 6
3111354.80255935 10162036.209444 3111456.389626510162033.9394354
3111507.6483822810162044.40037253111918.7656702710162102.4589834
3112168.7835429310162126.51930283112347.4360727710162146.7390786

Type RM Length L Ch R = 1 ,945.4837,78.84,84.39,89.94
XS GIS Cut Line= 2
3111407.2135437710162399.39474133111411.55408627 10161674.568435
#Sta/Elev= 30
       0  768.71   36.49  767.08   48.49  766.78  171.96  765.36  214.95  764.54
  226.45   764.5  233.95  764.05  239.45     764  256.44  762.43  316.93  755.16
   344.4  753.01  353.92  752.26  357.92  752.24  364.42  751.76  384.42  753.32
  390.41  753.83  391.41  754.05  399.41  757.01  404.41  758.03   448.9  759.89
   451.9  760.79   453.9  761.75   458.4  764.31   461.9  765.78   468.9   765.9
  493.89  767.46  539.38  769.34  546.38  768.92  634.86  769.99  724.84   770.4
#Mann= 1 ,-1 , 0
       0    .045       0
Bank Sta=344.4,384.42
XS Rating Curve= 0 ,0
Exp/Cntr=0.3,0.1

Type RM Length L Ch R = 1 ,861.0955,58.87,60.06,61.24
Node Name=WalshU
XS GIS Cut Line= 2
3111453.6547238510162378.56144963111533.5157845910161694.5336182
#Sta/Elev= 30
       0  767.82   19.99  766.95   26.49  766.23   55.97   766.3   63.47  765.64
   70.97  766.02  162.42  764.33   206.4  762.88  264.38  757.97  294.86  753.63
  306.86  754.05  319.36  753.21  320.35  753.23  322.85  754.37  337.34  754.21
  339.34  751.64  340.34   753.8  340.84  754.06  342.84   753.3  344.84  753.19
  359.51   754.2  374.82   754.1  389.32  756.63  398.81  758.78  406.31   759.5
   421.3   759.9   433.8  765.29  462.28  767.48  576.23  769.83  688.67  769.34
#Mann= 1 ,-1 , 0
       0    .045       0
Bank Sta=319.36,359.51
XS Rating Curve= 0 ,0
Exp/Cntr=0.3,0.1

Type RM Length L Ch R = 1 ,801.0373,81.01,81.04,81.07
XS GIS Cut Line= 2
3111505.7379530110162382.03388363111599.4880936110161715.3669098
#Sta/Elev= 30
       0  767.61  114.95  765.59  119.45   765.3  149.44  765.63  168.93  764.96
  182.43  763.77  193.92  762.46  198.42  762.56  261.39  758.69  280.89  757.21
  282.89  756.94  290.38  754.89  296.88  753.75  314.58  752.32  318.87  751.96
  323.87  751.19  354.58  750.97  357.35  750.83  379.85  752.86  382.84  753.41
  389.34  755.92  394.34  758.54  396.84  759.44  419.83  760.27  424.33  762.08
  427.83  764.16  433.32  766.35  437.82  766.78  578.26  769.59  673.23  769.41
#Mann= 1 ,-1 , 0
       0    .045       0
Bank Sta=314.58,354.58
XS Rating Curve= 0 ,0
Exp/Cntr=0.3,0.1

Type RM Length L Ch R = 1 ,719.9998,80,80,80
XS GIS Cut Line= 2
3111590.62131342 10162359.0946253111674.5217361710161764.9898421
#Sta/Elev= 30
       0  766.75   108.5  764.93     127  764.16     181  761.27   188.5  761.22
   201.5  760.63   213.5  759.65   224.5  758.62   244.5  756.46     250  755.42
     251  755.16     254  754.01     255  753.77     280  751.17     282     751
   300.5  750.95     320  751.75   327.5  752.07   343.5  754.17     350  755.84
     364  759.22   374.5  760.27     387  760.79   389.5  761.04     394  761.93
   397.5  763.32   401.5  764.72   403.5  765.26   411.5  766.14  600.01  769.21
#Mann= 1 ,-1 , 0
       0    .045       0
Bank Sta=280,320
XS Rating Curve= 0 ,0
Exp/Cntr=0.3,0.1

Type RM Length L Ch R = 1 ,640     ,80,80,80
XS GIS Cut Line= 2
3111669.8353938510162370.2812824 3111753.735816610161776.1764995
#Sta/Elev= 30
       0   767.1      18  766.92     144  763.51     147  763.11   191.5  761.11
     248  753.99     258  753.29   266.5  750.74     269   750.4     280   750.7
   300.5  750.73   309.5  750.44     320  752.04     326  750.99   327.5  750.94
     335  753.13   346.5   754.2   357.5  756.68     361  757.18   371.5  760.14
   382.5  760.98   398.5  761.69   415.5  763.51     428  764.46   437.5  764.91
   440.5  765.35     444  766.56     450   767.4     454  767.63  600.01  768.79
#Mann= 1 ,-1 , 0
       0    .045       0
Bank Sta=280,320
XS Rating Curve= 0 ,0
Exp/Cntr=0.3,0.1

Type RM Length L Ch R = 1 ,559.9999,80,80,80
XS GIS Cut Line= 2
3111749.0491461810162381.46826793111832.9495689310161787.3631569
#Sta/Elev= 30
       0  766.92   63.95  765.61  129.39  763.21  144.88  762.23  198.34  759.39
  231.31  756.93   239.8  755.63   240.8  755.35   245.3  752.95  248.29   752.1
  254.79  751.45  256.79   750.9  261.78  750.69     280  750.67  301.25  750.59
  315.24  751.49     320  752.04  323.73  752.46  336.72  752.65   357.7  756.75
   366.7  758.13  373.19  759.35  375.19  760.04  380.18  761.21  401.67  762.23
  412.16     765  425.15  766.16  428.14  766.56  522.07  767.87     600  768.07
#Mann= 1 ,-1 , 0
       0    .045       0
Bank Sta=280,320
XS Rating Curve= 0 ,0
Exp/Cntr=0.3,0.1

Type RM Length L Ch R = 1 ,479.9999,82.22,80,77.78
XS GIS Cut Line= 2
 3111828.263226610162392.65492533111912.1636493510161798.5498144
#Sta/Elev= 29
       0  766.34   71.94  765.87  105.91  765.27  138.88  762.64  216.82  758.43
  228.81  757.33   238.3  756.16  267.78  750.59  268.28  750.53     280  750.43
  300.75  750.47  308.74  751.35     320   751.1  324.73   750.9  326.23  751.04
  326.73  751.04  328.23  750.92  330.73  751.04  353.71  755.47   361.7  757.56
  377.19  760.33  390.68  761.87  391.18   761.9  404.16  762.02  406.16  762.28
  427.14  765.97  433.64  766.61  490.59   767.4     600  767.74
#Mann= 1 ,-1 , 0
       0    .045       0
Bank Sta=280,320
XS Rating Curve= 0 ,0
Exp/Cntr=0.3,0.1

Type RM Length L Ch R = 1 ,400.0002,80,80,80
XS GIS Cut Line= 2
 3111920.851624110162404.04565063111978.3269028410161806.8047191
#Sta/Elev= 30
       0   766.5   64.95  764.95  128.89  761.41  152.87  760.96  162.86  760.61
  191.84  760.45  203.33  759.83  214.82  758.29  230.31   757.6  262.28  752.32
  267.28  751.38  276.27  750.55     280  750.39  296.25  750.26  310.74  750.42
     320  750.14  325.73   750.1  335.72   751.2  337.72  751.66  341.22  752.02
  347.21  752.96   363.2  757.43  380.18  760.98  387.68  761.47  417.15  762.54
  421.65  763.31  438.63   765.3  462.11  766.76  471.11  767.05     600  767.39
#Mann= 1 ,-1 , 0
       0    .045       0
Bank Sta=280,320
XS Rating Curve= 0 ,0
Exp/Cntr=0.3,0.1

Type RM Length L Ch R = 1 ,319.9999,80,80,80
XS GIS Cut Line= 2
3112000.4840107610162411.70902113112057.9589614310161814.4680896
#Sta/Elev= 30
       0  766.32   18.48   766.6   64.95  765.51  110.91  761.68  158.37  759.59
  181.35  758.09  222.31  756.14  227.81  756.09   243.8  753.53  249.79  752.01
  268.78  750.24     280   750.2  284.76  750.13  290.76  750.74  298.25  750.63
  300.25  750.21  304.75  750.99     320  750.88  327.73  750.87  330.72  751.14
  346.21  754.56  351.21  755.96  365.69  758.67  374.19   759.5  398.67  761.31
  415.15  762.19  418.15  762.78  440.13  765.44  456.12  766.35     600  766.97
#Mann= 1 ,-1 , 0
       0    .045       0
Bank Sta=280,320
XS Rating Curve= 0 ,0
Exp/Cntr=0.3,0.1

Type RM Length L Ch R = 1 ,240     ,79.16,80,80.84
XS GIS Cut Line= 2
3112080.1160693510162419.37239163112137.5910200210161822.1314601
#Sta/Elev= 30
       0  765.61   35.97  765.63   55.45  765.35   64.45  765.59   76.94  764.84
  126.89  760.74  161.37  759.22  183.35  758.88  200.33  757.89  209.33  757.17
   240.8  754.14  248.79  753.06  262.78  750.74  266.28  750.49     280  750.19
  310.24  750.13     320  750.72  334.72  751.72  347.21  754.72  351.71  755.97
   364.7  758.56  382.18  760.04  385.18  760.12  394.67  760.84  416.15  761.83
  444.63  764.99  448.12  765.12  455.62  766.59   472.1  766.27     600  766.38
#Mann= 1 ,-1 , 0
       0    .045       0
Bank Sta=280,320
XS Rating Curve= 0 ,0
Exp/Cntr=0.3,0.1

Type RM Length L Ch R = 1 ,159.9999,120,120,120
XS GIS Cut Line= 2
3112154.7127049310162426.8421929 3112222.189604110161830.6485034
#Sta/Elev= 25
       0  765.64   65.45  765.32   70.94  765.05   120.9  760.97  133.39   760.1
  218.32  755.57  269.78   750.1     280  749.93  312.74     750     320  750.71
  338.22  752.44  341.22   752.9  344.71  753.88  349.71     756   361.7  758.31
  382.68  759.94  399.17  760.74  415.15  761.13  421.15  761.83  432.14  764.59
  433.14  764.72  439.63  764.97   474.6  765.77  519.56  766.09     600  765.99
#Mann= 1 ,-1 , 0
       0    .045       0
Bank Sta=280,320
XS Rating Curve= 0 ,0
Exp/Cntr=0.3,0.1

Type RM Length L Ch R = 1 ,40.00006,40,40,40
XS GIS Cut Line= 2
3112273.9513115910162440.33757283112341.4282107710161844.1438833
#Sta/Elev= 30
       0  764.99   69.94  764.24   86.93  761.82   120.4  759.38   237.3  753.83
   246.8  751.22  259.78  749.44     280  749.56  297.75  749.74  299.75  749.39
  306.25  750.79     320  750.41  335.22  751.88  342.21  753.61  366.19  752.62
  382.18  753.05  384.68  753.98  390.17  757.61  395.17  760.14  414.65  760.51
  422.65  758.26  424.14  758.48  426.64  757.75  432.14  757.51  440.63  761.69
  449.62  763.73  462.11  764.82  505.08  766.44  555.53   765.6     600  765.88
#Mann= 1 ,-1 , 0
       0    .045       0
Bank Sta=280,320
XS Rating Curve= 0 ,0
Exp/Cntr=0.3,0.1

Chan Stop Cuts=-1
Use User Specified Reach Order=0
Composite Channel Slope=5
